--- SrvyrCrk.prj (project) ---

Proj Title=SrvyrCrk
Current Plan=p01
Default Exp/Contr=0,0
English Units
Geom File=g01
Flow File=f01
Plan File=p01
BEGIN DESCRIPTION:
END DESCRIPTION:
DSS Export Rating Curves= 0
DSS Export Rating Curve Sorted= 0
DSS Export Volume Flow Curves= 0
DXF OffsetX= 0
DXF OffsetY= 0
DXF ScaleX= 0
DXF ScaleY= 0

--- SrvyrCrk.p01 (plan) ---

Plan Title=Floodplain
Program Version=4.00
Geom File=g01
Flow File=f01
K Sum by GR=0
Std Step Tol=0.01
Critical Tol=0.01
Num of Std Step Trials=20
Max Error Tol=0.3
Flow Tol Ratio=0.001
Split Flow NTrial=30
Split Flow Tol=0.02
Split Flow Ratio=0.02
Log Output Level=0
Friction Slope Method=1
Unsteady Friction Slope Method=2
Unsteady Bridges Friction Slope Method=1
Global Log Level=0
CheckData=False
Run HTab=0
Run UNet=0
Run PostProcess=0
UNET Theta=0
UNET Theta Warmup=0
UNET ZTol=0
UNET ZSATol=0
UNET MxIter=0
UNET MaxInSteps=0
UNET DtIC=0
UNET DtMin=0
UNET MaxCRTS=0
UNET WFStab=0
UNET SFStab=0
UNET WFX=0
UNET SFX=0
UNET DSS MLevel=0
UNET DZMax Abort=0
UNET Convert EG Bridges=0
UNET Use Existing IB Tables=0
UNET Froude Limit=0
UNET Froude Power=0
Write IC File=0
Echo Input=False
Echo Output=False
Write Detailed=0

--- SrvyrCrk.f01 (steady flow) ---

Flow Title=NFF Regression Equation
Program Version=4.00
Number of Profiles=1
Profile Names=P100yr
River Rch & RM=SrvyrCrk,Main      ,17560.4
885.6909
River Rch & RM=SrvyrCrk,Main      ,17120.7
897.6510
River Rch & RM=SrvyrCrk,Main      ,16625.6
1082.475
River Rch & RM=SrvyrCrk,Main      ,14995.8
1133.620
River Rch & RM=SrvyrCrk,Main      ,14781.2
1263.216
River Rch & RM=SrvyrCrk,Main      ,11285
1345.312
River Rch & RM=SrvyrCrk,Main      ,10982.9
1505.011
River Rch & RM=SrvyrCrk,Main      ,10629.7
1518.907
River Rch & RM=SrvyrCrk,Main      ,5483.3
1678.975
River Rch & RM=SrvyrCrk,Main      ,4249.7
1834.080
River Rch & RM=SrvyrCrk,Main      ,258.5
1972.907
Boundary for River Rch & Prof#=SrvyrCrk,Main      ,1
Up Type=0
Dn Type=3
Dn Slope=0.008555

--- SrvyrCrk.g01 (geometry) ---

Geom Title=USGS 3m DEM
Program Version=4.10

River Reach=SrvyrCrk        ,Main
Reach XY= 30
     1880740.342      265591.081      1881365.76      267645.547
     1881343.207      268456.967     1881188.259      268690.039
     1880823.676      268910.091     1880309.466      269570.135
     1880354.926      269735.612     1879904.405      270618.425
     1880002.061      270936.133     1879962.619      271223.811
     1880134.915      271282.887     1880255.967      271552.019
     1880047.634      271674.415     1879986.841      272447.775
     1879744.248      272654.883     1879485.134      273100.196
     1879104.237      273525.346      1878573.71      274001.219
     1878555.304      274390.024     1878265.082      274662.696
     1878250.662      274932.514     1878336.696      275128.841
     1878279.891      275284.482     1877673.936      275318.946
     1877156.266      275871.085     1876469.509      278282.487
     1876505.967      278485.612     1876352.913      279250.632
     1875890.322      279230.942     1875673.701      279668.419

Type RM Length L Ch R = 1 ,17560.4 ,440.8,439.7,438.6
XS GIS Cut Line= 2
     1880003.607      265817.263     1881657.141      265349.541
#Sta/Elev= 30
       0 2057.03      30 2055.17   189.8 2049.17   209.8 2046.32   239.8 2043.17
   319.7 2037.64   359.7 2034.34   369.7 2032.89   399.6 2032.97   419.6 2035.86
   439.6 2036.76   489.6 2036.64   549.5 2037.27   599.4 2036.69   699.4 2038.35
   719.3 2036.49   739.3 2033.33   760.5 2032.59   780.5  2032.6   859.2 2033.65
   909.2 2033.67    1069  2031.8  1158.9 2032.21  1328.8  2035.5  1358.7 2037.14
  1428.7 2039.65  1578.5 2044.17  1638.5 2046.94  1668.5 2047.63  1718.4 2050.24
#Mann= 3 , 0 , 0
       0     .06       0   760.5    .045       0   780.5     .06       0
#XS Ineff= 2 , 0
          434.29 2036.76
Permanent Ineff=
       F       F
Bank Sta=760.5,780.5
XS Rating Curve= 0 ,0
Exp/Cntr=0.3,0.1

Type RM Length L Ch R = 1 ,17120.7 ,137.6,138.1,138.7
XS GIS Cut Line= 2
     1880335.334       266203.78     1881618.622      265781.496
#Sta/Elev= 30
       0  2052.1      20 2053.02      40 2055.01    80.1 2055.35   150.1 2053.13
   300.2 2052.13   310.2 2050.54   350.2 2034.96   360.3 2032.37   380.3 2031.53
   490.4  2033.6   544.3  2029.8   550.4  2029.7   564.3  2029.7   790.6 2033.79
   860.6 2033.32   990.7 2030.51  1010.7 2030.53  1080.8 2032.82  1100.8 2034.73
  1110.8 2037.39  1120.8 2040.68  1140.8 2048.69  1180.9 2060.58  1190.9    2065
  1200.9 2068.45  1220.9 2070.97  1260.9  2073.4  1280.9 2075.55    1351 2080.38
#Mann= 3 , 0 , 0
       0     .06       0   544.3    .045       0   564.3     .06       0
Bank Sta=544.3,564.3
XS Rating Curve= 0 ,0
Exp/Cntr=0.3,0.1

Type RM Length L Ch R = 1 ,16982.6 ,357.2,356.9,356.6
XS GIS Cut Line= 2
     1880375.669      266323.863     1881596.612      265949.326
#Sta/Elev= 30
       0 2054.29    29.9 2054.05    49.9 2052.43    69.8 2052.68   139.7 2056.19
   169.6 2058.58   189.6 2059.03   219.5 2058.42   229.5 2057.98   309.3 2050.18
   319.3 2048.02   329.2 2041.69   349.2 2033.56   359.2 2030.99   369.2 2030.12
   498.9 2033.03     536 2031.17     556 2029.78   578.7 2029.57   718.4  2030.9
   818.1 2033.09  1027.7    2036  1107.5    2038  1117.5  2039.2  1127.4 2041.82
  1147.4 2049.61  1157.4 2055.87  1187.3 2065.33  1227.2 2072.75  1277.1 2076.63
#Mann= 3 , 0 , 0
       0     .06       0     536    .045       0     556     .06       0
Bank Sta=536,556
XS Rating Curve= 0 ,0
Exp/Cntr=0.3,0.1

Type RM Length L Ch R = 1 ,16625.6 ,360.6,361,361.5
XS GIS Cut Line= 2
     1880474.977      266673.248     1881893.753      266218.953
#Sta/Elev= 30
       0 2042.67      20 2041.85      50 2039.48      60 2039.56      80 2042.43
     100  2047.5     110 2047.97     120 2044.89     130 2040.78     140 2038.93
     180 2038.66     250 2035.72   309.9 2033.82   379.9 2034.18   459.9 2033.64
   519.9 2034.41   529.9 2034.12   549.9 2030.81   561.3 2029.39   569.9 2029.26
   589.9 2029.42   749.9 2030.59  1019.8 2030.96  1139.8 2034.04  1199.8 2035.06
  1239.8  2035.2  1289.8 2037.19  1319.8 2039.87  1379.8 2041.95  1489.7 2049.52
#Mann= 3 , 0 , 0
       0     .06       0   561.3    .045       0   589.9     .06       0
Bank Sta=561.3,589.9
XS Rating Curve= 0 ,0
Exp/Cntr=0.3,0.1

Type RM Length L Ch R = 1 ,16264.4 ,194.9,193.2,191.5
XS GIS Cut Line= 3
     1880501.593      266997.572     1880823.496      266934.292
     1881731.426      266661.913
#Sta/Elev= 30
       0 2057.02    39.8 2051.83    49.7 2049.78   139.2 2039.64   159.1 2039.14
   198.8 2040.17   278.4 2045.36   288.3 2045.15   318.1 2039.07     338 2036.29
     378 2031.84   397.9  2030.8   447.8 2030.55   597.5 2035.57   607.4 2035.48
   628.1 2030.31   637.4 2029.27   647.4  2029.2   648.1 2029.21     817 2029.64
   956.7 2034.77  1036.5 2033.31  1056.4 2033.81  1106.3  2043.6  1116.3 2047.44
  1176.2  2060.7  1196.2 2066.81  1226.1 2070.01    1266 2072.41    1276 2073.92
#Mann= 3 , 0 , 0
       0     .06       0   628.1    .045       0   648.1     .06       0
#XS Ineff= 2 , 0
          599.53 2035.64
Permanent Ineff=
       F       F
Bank Sta=628.1,648.1
XS Rating Curve= 0 ,0
Exp/Cntr=0.3,0.1

Type RM Length L Ch R = 1 ,16071.1 ,299.4,300,300.7
XS GIS Cut Line= 3
     1880675.904      267217.576     1881188.342       267025.82
     1881698.966      266833.635
#Sta/Elev= 30
       0 2056.45    49.7 2053.72   149.2  2052.7   179.1 2051.37     199 2048.88
   258.6  2037.9   268.6 2036.48   278.5 2035.89   507.4 2035.37   517.3 2034.96
   537.1  2030.8   547.1 2028.84   557.1 2028.99   576.9 2029.95   606.7 2030.41
   715.8 2030.09   854.7 2035.52   864.6 2035.65   874.5 2035.19   884.4 2033.94
   894.3 2033.78   904.3 2034.93   914.2 2037.51   943.9 2049.39   953.9 2052.59
   963.8 2056.87   973.7 2059.52  1043.1 2073.22    1053 2075.99  1092.7 2079.63
#Mann= 3 , 0 , 0
       0     .06       0   537.1    .045       0   557.1     .06       0
Bank Sta=537.1,557.1
XS Rating Curve= 0 ,0
Exp/Cntr=0.3,0.1

Type RM Length L Ch R = 1 ,15771.1 ,326.5,327.2,327.9
XS GIS Cut Line= 3
     1880762.837      267490.249     1881278.847      267311.784
     1881794.857      267133.319
#Sta/Elev= 30
       0 2098.87    39.7 2092.34    49.6 2089.67    79.4 2084.14   109.2 2077.22
     129 2070.23   198.6 2054.04   208.5  2049.9   287.9 2033.85   297.8 2032.44
   367.3 2031.88   516.2 2034.18   526.2 2032.99     536 2029.94     546 2026.54
   555.9 2026.36     556 2026.36   724.7 2029.83   784.2 2032.11   873.6  2036.8
   883.5 2038.12   893.4 2041.65   913.3 2051.37   923.2 2054.98     953 2062.08
     963 2065.48  1032.4 2079.31  1042.4 2081.88  1072.2 2086.57    1092 2091.56
#Mann= 3 , 0 , 0
       0     .06       0     536    .045       0     556     .06       0
Bank Sta=536,556
XS Rating Curve= 0 ,0
Exp/Cntr=0.3,0.1

Type RM Length L Ch R = 1 ,15443.9 ,439.5,448.1,456.7
XS GIS Cut Line= 3
     1880812.429      267681.169      1881107.31      267707.451
     1882059.089      267408.763
#Sta/Elev= 30
       0 2092.32    29.6 2088.22    39.5 2085.31      79 2066.68     148 2048.86
   157.9 2045.56   167.8 2044.25   197.4 2041.79   246.7 2041.58   385.8 2035.55
   525.5 2032.73   545.4 2030.44   565.4  2025.8   575.4 2025.78   585.3 2025.83
     715  2026.3   904.6 2038.92   934.5 2038.44   974.4 2033.11   994.3 2033.24
  1024.3 2035.19  1054.2 2040.92  1094.1 2046.41  1104.1 2047.03    1124 2047.44
    1144 2045.35  1183.9  2044.9  1223.8 2046.54  1263.7 2049.56  1293.6 2045.94
#Mann= 3 , 0 , 0
       0     .06       0   565.4    .045       0   585.3     .06       0
Bank Sta=565.4,585.3
XS Rating Curve= 0 ,0
Exp/Cntr=0.3,0.1

Type RM Length L Ch R = 1 ,14995.8 ,213.1,214.5,216
XS GIS Cut Line= 3
     1880911.318      268057.868     1881741.829      268088.163
     1882203.016      268102.092
#Sta/Elev= 30
       0 2083.95    49.5 2077.26    59.4 2074.99    69.3 2069.92    79.2  2067.9
    98.9 2065.21   138.5 2062.14   148.4 2058.54   227.6 2039.66   306.7 2030.24
   336.4 2029.64   405.6  2031.4   425.4    2030     445 2025.91     465  2024.6
   573.8 2027.02   821.2 2028.66   850.7 2029.42   899.8  2033.3   929.2 2036.28
   948.9 2039.44  1007.8 2043.94  1066.7 2049.87  1145.2 2061.96  1164.8 2065.87
  1184.5 2072.73  1233.6 2083.32  1253.2  2089.9    1263 2095.46  1292.5 2101.96
#Mann= 3 , 0 , 0
       0     .06       0     445    .045       0     465     .06       0
Bank Sta=445,465
XS Rating Curve= 0 ,0
Exp/Cntr=0.3,0.1

Type RM Length L Ch R = 1 ,14781.2 ,221.7,232.3,243
XS GIS Cut Line= 3
     1880864.183      268241.729     1881407.733      268293.476
     1881951.021      268347.805
#Sta/Elev= 30
       0 2118.45    29.8 2109.88    39.7 2105.93    49.6 2101.41   109.2 2084.28
   119.1 2080.76   129.1 2076.08   188.6 2059.78   198.6 2056.65   208.5 2051.76
   248.2 2040.89   258.1 2039.01     278 2037.28   347.5  2033.6   357.4 2032.59
   377.2 2031.47     407 2030.47   426.9 2029.33   436.8  2027.9   482.1 2023.53
   496.4 2022.42   502.1 2022.37   506.3 2022.33   526.2 2023.71   595.6 2026.59
   903.4 2032.14   982.8 2034.61  1032.4 2036.87  1072.2 2037.67    1092 2038.72
#Mann= 3 , 0 , 0
       0     .06       0   482.1    .045       0   502.1     .06       0
Bank Sta=482.1,502.1
XS Rating Curve= 0 ,0
Exp/Cntr=0.3,0.1

Type RM Length L Ch R = 1 ,14548.8 ,309.1,318.6,328.1
XS GIS Cut Line= 3
     1880801.408       268250.82     1881050.048       268362.09
     1881784.899      268781.336
#Sta/Elev= 30
       0 2136.96    19.5 2133.13    29.2 2128.89     107 2104.59   116.7 2099.64
   194.6 2073.65   204.3 2068.36   282.4  2043.5   292.3 2038.81   302.3 2036.46
   401.8  2031.2   461.5  2029.4   501.3 2026.96   551.1 2022.74     561 2021.89
     571 2021.95   590.9 2026.82   620.8 2028.42   650.6 2031.69   670.5 2035.17
   740.2 2044.38   770.1 2049.36   809.9 2054.52   839.7 2056.88   859.6 2060.04
   929.3 2071.67    1009 2087.55  1058.7 2096.11  1088.6 2103.69  1118.4 2110.22
#Mann= 3 , 0 , 0
       0      .1       0   551.1    .045       0     571      .1       0
Bank Sta=551.1,571
XS Rating Curve= 0 ,0
Exp/Cntr=0.3,0.1

Type RM Length L Ch R = 1 ,14230.2 ,412.1,408.8,408.5
XS GIS Cut Line= 2
     1880749.586      268318.723     1881462.996      269159.591
#Sta/Elev= 30
       0  2128.4     9.9 2127.38    19.9 2125.01    79.5 2104.57   119.2 2092.52
   129.2  2089.8     149 2087.61     159  2084.9   228.5 2062.63   258.3  2050.7
   278.2 2046.59     308 2036.48   317.9 2034.69   327.8 2034.11   476.9 2028.69
   547.1 2021.74   566.3 2021.13   567.1 2021.21   615.9 2028.72   705.4 2030.21
   725.2 2031.98   735.2 2033.86   774.9 2045.59   844.4 2053.46     904 2064.24
   923.9 2065.86   983.5 2075.48  1033.2 2086.82  1053.1 2088.68  1102.7 2097.82
#Mann= 3 , 0 , 0
       0      .1       0   547.1    .045       0   567.1      .1       0
Bank Sta=547.1,567.1
XS Rating Curve= 0 ,0
Exp/Cntr=0.3,0.1

Type RM Length L Ch R = 1 ,13821.4 ,155.5,152,149.9
XS GIS Cut Line= 2
     1880571.837      268702.564     1881206.669      269371.387
#Sta/Elev= 30
       0 2066.76     9.9 2066.13    39.7  2058.3    49.6 2057.58     119 2040.04
   138.8 2036.02   330.7 2019.84     347 2019.08   350.7 2019.49     357  2020.2
   376.8 2027.12   386.7 2028.07   436.3 2028.35   446.2 2029.62     466 2034.27
   485.9  2035.7   495.8 2037.46   525.5 2048.52   545.4 2053.41   565.2  2056.2
   614.8 2068.74   634.6 2075.11   664.3 2083.28   694.1 2088.66   803.2 2119.33
   813.1 2121.65     823 2122.52   842.8 2128.39   872.6 2134.15   922.1 2151.32
#Mann= 3 , 0 , 0
       0      .1       0   330.7    .045       0   350.7      .1       0
Bank Sta=330.7,350.7
XS Rating Curve= 0 ,0
Exp/Cntr=0.3,0.1

Type RM Length L Ch R = 1 ,13669.4 ,302.4,300,297.4
XS GIS Cut Line= 3
     1880299.029       268724.87     1880719.352       269073.97
     1881124.804       269439.57
#Sta/Elev= 30
       0 2072.03    29.8 2069.48   119.2 2056.48   139.1  2054.8   208.6 2041.56
     298 2037.02   407.3 2027.28   536.4 2019.13   546.4 2019.47   556.4 2021.78
   566.2 2025.36   576.2  2027.4     596 2028.96   615.9 2034.52   635.7 2038.52
   655.6  2039.7   665.5 2041.64   685.4  2050.1   725.1 2064.05     735 2065.02
   794.6 2079.06   824.3  2087.7     864 2100.65   883.9 2103.48   933.5 2117.28
    1003 2139.17  1022.8 2142.03  1042.7 2149.03  1062.6  2158.4  1092.3 2170.57
#Mann= 3 , 0 , 0
       0      .1       0   536.4    .045       0   556.4      .1       0
Bank Sta=536.4,556.4
XS Rating Curve= 0 ,0
Exp/Cntr=0.3,0.1

Type RM Length L Ch R = 1 ,13369.4 ,282.6,285.6,287.8
XS GIS Cut Line= 3
     1880073.526      268995.596     1880525.077      269302.418
     1880966.033      269625.086
#Sta/Elev= 30
       0 2064.73    69.5 2058.22     129 2058.11   158.8 2053.62   178.7 2048.18
   208.4  2042.9   277.9 2033.85   377.2 2028.95     407 2028.41   476.4    2022
   535.9 2019.38   545.9 2018.86   555.9 2019.01   585.7 2025.88   605.5 2028.59
   625.4 2033.73   645.3 2034.99   665.1 2040.59   744.6 2058.73   764.5 2065.36
     844 2082.78   863.8 2089.78   943.3 2110.96   963.2  2118.2   973.1 2123.27
  1012.9 2133.71  1052.6 2145.64  1062.5 2149.15  1072.5 2154.36  1092.3 2160.16
#Mann= 3 , 0 , 0
       0     .06       0   535.9    .045       0   555.9     .06       0
Bank Sta=535.9,555.9
XS Rating Curve= 0 ,0
Exp/Cntr=0.3,0.1

Type RM Length L Ch R = 1 ,13083.8 ,320.7,317.5,314.2
XS GIS Cut Line= 3
     1879945.952      269172.359     1880469.695      269631.128
     1880902.382      269721.457
#Sta/Elev= 30
       0  2123.1    19.9  2118.7    29.8 2114.45   119.4 2098.37   159.1 2087.66
   208.9 2078.37   238.7  2069.1   258.6 2059.84   288.4 2049.98   348.1 2038.85
   387.9 2040.18   417.8 2038.42   487.4 2024.67   529.5 2019.71   547.1 2018.29
   549.5 2018.43   596.8 2024.47   666.4 2026.63   715.9 2031.95   745.4 2033.02
     765 2035.96   843.6 2052.99   863.2 2059.14     932 2075.59   941.8 2080.73
  1010.6 2100.27  1030.2 2108.82  1089.2    2128  1108.8 2138.17  1138.3 2148.46
#Mann= 3 , 0 , 0
       0     .06       0   529.5    .045       0   549.5     .06       0
Bank Sta=529.5,549.5
XS Rating Curve= 0 ,0
Exp/Cntr=0.3,0.1

Type RM Length L Ch R = 1 ,12766.2 ,298.6,293.5,288.4
XS GIS Cut Line= 3
     1879756.209      269679.468     1880184.935       269720.89
     1880766.676      270093.575
#Sta/Elev= 30
       0 2162.75    58.7 2141.76    78.3 2131.55     137 2111.45   156.6 2102.24
   225.2 2081.91   234.9 2077.06   303.5 2058.93   313.2 2054.65   381.8 2040.06
   411.1 2033.03   430.7 2031.17   460.3  2026.4   564.5 2019.58   578.8 2018.26
   584.5 2018.34     638 2024.29   667.6 2025.52   726.8 2031.36     786 2035.52
     865 2048.58   874.9 2051.77   953.8 2069.45   973.6  2076.2  1003.2 2083.98
  1022.9    2092  1052.5 2102.66  1062.4 2109.23  1072.2  2114.5  1121.6 2136.77
#Mann= 3 , 0 , 0
       0     .06       0   564.5    .045       0   584.5     .06       0
Bank Sta=564.5,584.5
XS Rating Curve= 0 ,0
Exp/Cntr=0.3,0.1

Type RM Length L Ch R = 1 ,12472.7 ,293.8,300,303.4
XS GIS Cut Line= 3
     1879680.174      269869.782     1880189.458      270066.612
     1880698.822      270263.256
#Sta/Elev= 30
       0  2130.1    69.5 2108.31    89.3  2100.3   158.8 2083.03   168.8 2076.64
   198.5 2062.52   228.3 2053.13   238.2 2051.51     278 2049.76   317.7 2043.92
   327.6 2042.08   347.4 2035.71   416.9 2020.78     536 2012.47     546 2012.06
     556 2012.21   605.6 2014.06   655.2 2022.11   794.2 2034.53     814 2038.26
   853.7    2054   863.7  2060.7   873.6 2065.11   923.2 2068.79   943.1 2073.73
     953 2078.59  1002.6 2096.28  1022.5 2104.69  1042.4 2116.46    1092 2139.94
#Mann= 3 , 0 , 0
       0      .1       0     536    .045       0     556      .1       0
Bank Sta=536,556
XS Rating Curve= 0 ,0
Exp/Cntr=0.3,0.1

Type RM Length L Ch R = 1 ,12172.7 ,268.6,258.6,251.4
XS GIS Cut Line= 3
     1879616.064      270020.451     1880063.113      270337.013
     1880544.736      270603.246
#Sta/Elev= 30
       0 2145.02    59.8 2126.71    79.7  2118.3   159.4 2096.57     259 2059.98
   278.9 2049.29   308.8  2038.9   328.7 2033.72   368.5 2020.82   378.5 2018.64
   408.4 2016.93   458.1  2007.6   537.8 2002.04   557.8 2002.71   637.8 2003.45
   657.8 2004.94   667.8 2009.98   687.9 2012.68   707.9 2017.57   737.9 2021.38
   757.9 2025.95   777.9 2032.83   807.9 2039.54   837.9 2045.58     858 2047.51
     938 2065.47     978 2085.96    1028 2106.76  1048.1 2117.17  1098.1 2130.89
#Mann= 3 , 0 , 0
       0      .1       0   537.8    .045       0   557.8      .1       0
Bank Sta=537.8,557.8
XS Rating Curve= 0 ,0
Exp/Cntr=0.3,0.1

Type RM Length L Ch R = 1 ,11914.1 ,353.1,341.4,330.8
XS GIS Cut Line= 3
     1879420.897      270385.798      1879858.39      270539.575
     1880509.622      270681.507
#Sta/Elev= 30
       0 2116.34    19.7  2117.4    39.5  2116.3    88.8 2109.42     148 2092.61
   217.1 2067.62   325.6 2038.32   384.8  2017.3   434.1 2014.01     444 2011.12
   463.7  2001.2   483.6 1995.52   528.8 1993.19   548.8  1992.8   553.3 1992.79
     603 1993.54   712.4 2001.68   752.2 2009.56   782.1  2017.5   811.9  2020.3
   861.6 2035.06   881.6 2043.75   911.4 2046.66   931.3 2050.94   961.1 2063.13
  1020.8 2081.88  1040.7 2090.74  1110.4 2110.26  1120.3 2115.84  1130.2 2118.59
#Mann= 3 , 0 , 0
       0     .08       0   528.8    .045       0   548.8     .08       0
Bank Sta=528.8,548.8
XS Rating Curve= 0 ,0
Exp/Cntr=0.3,0.1

Type RM Length L Ch R = 1 ,11572.7 ,283.6,287.6,290.3
XS GIS Cut Line= 3
     1879419.049      271003.842     1879952.582      270874.821
     1880514.804      270763.701
#Sta/Elev= 30
       0 2012.99   129.7  2012.1   179.6 2009.99   209.6 2009.69   259.5 2002.89
   299.4  2001.2   369.3  2001.2   379.2 2002.11   399.2 2007.15   409.2 2007.39
   469.1 1998.82   538.9  1992.5   558.9 1992.63   598.3 1993.93   637.8 1997.51
   687.2 1999.86   766.3  2013.3     786 2014.72   795.9 2016.46   855.2 2033.25
     875 2041.76   884.9 2044.22   914.5 2046.57   924.4 2048.81   944.2 2055.78
     954 2061.93  1023.2 2080.03  1033.1 2084.11  1092.4 2099.88    1122 2110.87
#Mann= 3 , 0 , 0
       0     .08       0   538.9    .045       0   558.9     .08       0
Bank Sta=538.9,558.9
XS Rating Curve= 0 ,0
Exp/Cntr=0.3,0.1

Type RM Length L Ch R = 1 ,11285   ,314.2,302.1,289.9
XS GIS Cut Line= 3
     1879411.131       271183.38     1880342.791      271095.166
     1880543.757      270921.302
#Sta/Elev= 30
       0 2078.87    49.8  2074.1   149.3 2056.08   209.1 2049.53     229 2045.44
   238.9 2046.71   258.8 2043.67   288.7 2038.59   298.7 2035.32   368.4 2020.82
   378.3 2017.54     448 2008.48   497.8 1994.23   544.5 1991.53   557.5 1991.27
   564.5 1991.47   627.2 1997.02   746.7  2000.1   776.5 2003.77   796.4 2009.94
   806.4 2011.58   925.9 2017.83     985  2024.9  1014.6 2030.28  1034.2 2036.17
  1063.8 2040.02    1113 2051.06  1142.5 2061.12  1162.2 2070.27  1201.6 2082.32
#Mann= 3 , 0 , 0
       0      .1       0   544.5    .045       0   564.5      .1       0
Bank Sta=544.5,564.5
XS Rating Curve= 0 ,0
Exp/Cntr=0.3,0.1

Type RM Length L Ch R = 1 ,10982.9 ,332.1,353.2,374.4
XS GIS Cut Line= 3
     1879516.156      271509.447     1880022.436      271372.188
     1880599.045       271028.84
#Sta/Elev= 30
       0 2146.81    39.6 2135.11    59.4 2125.82   118.8 2102.96   138.6 2091.25
   168.2 2079.87     198 2070.24   217.7  2061.8   277.1 2046.62   296.9  2039.2
   366.2 2022.09   376.1 2017.34   415.7 2007.58   425.6 2005.94   475.1 2004.06
   544.3 1998.28   623.2  1997.5   660.5 1990.88   662.7 1990.51   680.5 1991.68
   721.9 1995.23   781.2  2011.1   820.6 2012.37   840.4 2014.83   879.8 2024.63
   919.3  2032.4   978.5 2034.79  1047.6  2040.9  1185.8 2070.14  1195.6 2071.21
#Mann= 3 , 0 , 0
       0      .1       0   660.5    .045       0   680.5      .1       0
Bank Sta=660.5,680.5
XS Rating Curve= 0 ,0
Exp/Cntr=0.3,0.1

Type RM Length L Ch R = 1 ,10629.7 ,297.5,288.2,278.9
XS GIS Cut Line= 3
     1879535.433      271584.081     1880028.627      271539.329
     1880716.099      271789.253
#Sta/Elev= 30
       0 2152.55    19.8 2145.43    39.6 2134.28      99 2112.48   118.8 2100.29
   168.4 2075.03   217.9 2063.53   257.5 2050.27   277.3 2041.77   336.8 2026.49
   346.6 2022.25   425.9 2003.06   495.2 2000.44   633.6 1990.01   689.1 1989.71
   702.8 1989.58   709.1 1989.66   722.6 1991.42     772 2006.29   811.5 2008.28
   841.2    2013   900.5 2028.77   930.2  2038.5     940 2043.88   949.9 2046.91
   989.5    2050  1019.1 2057.45    1029 2061.97  1137.8 2082.75  1226.7 2093.52
#Mann= 3 , 0 , 0
       0      .1       0   689.1    .045       0   709.1      .1       0
Bank Sta=689.1,709.1
XS Rating Curve= 0 ,0
Exp/Cntr=0.3,0.1

Type RM Length L Ch R = 1 ,10341.5 ,243.1,250.2,257.3
XS GIS Cut Line= 3
     1879517.078      271773.107     1880225.173      271754.447
     1880611.056      271989.868
#Sta/Elev= 30
       0  2177.6    39.9 2161.69    49.9 2154.44    59.9 2149.65   119.7 2126.41
   139.7 2115.49   199.5  2094.9   219.5 2084.87   279.4  2065.4   299.3 2055.99
   359.2 2037.57   379.1 2028.34     439 2009.74     449 2004.85   458.9 2002.28
   488.8 2002.79   508.8 2000.94   528.8 1991.91   541.3 1989.42   548.7  1989.4
   561.3 1989.63   668.4 1996.04   796.8 2006.68   875.4 2017.87     895 2022.75
   963.8 2030.95   983.5 2036.73  1042.4 2046.49  1101.4 2050.39  1160.4 2056.89
#Mann= 3 , 0 , 0
       0      .1       0   541.3    .045       0   561.3      .1       0
Bank Sta=541.3,561.3
XS Rating Curve= 0 ,0
Exp/Cntr=0.3,0.1

Type RM Length L Ch R = 1 ,10091.3 ,217.4,213.4,209.4
XS GIS Cut Line= 2
     1879500.263      271861.152     1880581.241      272143.644
#Sta/Elev= 30
       0 2178.85    69.8 2150.31    79.8 2143.62   149.6 2115.32   169.6 2103.59
   199.5 2092.23   229.4 2082.32   249.4 2072.01   319.2  2050.5   329.2 2044.63
     399 2023.89     419 2015.99   468.9 2003.24   488.8  1999.6   518.7 1998.12
   566.5 1989.98   568.6  1989.7   586.5 1990.89   668.4 1997.25   788.1 2004.41
     818 2007.89     828 2010.56     838 2015.16   847.9 2017.75   947.7 2037.33
   987.6 2048.81  1017.5 2051.71  1057.4 2060.86  1077.4 2066.84  1117.3 2073.23
#Mann= 3 , 0 , 0
       0      .1       0   566.5    .045       0   586.5      .1       0
Bank Sta=566.5,586.5
XS Rating Curve= 0 ,0
Exp/Cntr=0.3,0.1

Type RM Length L Ch R = 1 ,9877.8  ,508,525.9,543.5
XS GIS Cut Line= 2
      1879437.05      272111.357     1880562.552      272268.253
#Sta/Elev= 30
       0 2170.12    59.8 2144.51    69.8 2137.76    79.8 2132.89   139.6 2109.41
   159.5 2098.19   209.3 2080.53   229.3 2071.38   289.1    2052     309 2042.19
   348.9 2027.04   388.8  2013.9   488.4 1996.53   508.4 1990.82   520.7 1988.66
   528.3 1988.28   540.7 1988.44   608.1 1991.25   717.7 2000.91   757.6 2002.34
   777.5  2004.6   807.4 2012.63   867.2 2025.18     957 2052.56   986.9 2055.69
  1026.7 2065.48  1046.7 2073.21  1106.5 2090.41  1126.4 2098.83  1136.4 2101.73
#Mann= 3 , 0 , 0
       0      .1       0   520.7    .045       0   540.7      .1       0
Bank Sta=520.7,540.7
XS Rating Curve= 0 ,0
Exp/Cntr=0.3,0.1

Type RM Length L Ch R = 1 ,9352    ,242.6,238.8,232.9
XS GIS Cut Line= 3
     1879336.827      272250.054     1879725.296       272483.37
     1880154.739      272973.845
#Sta/Elev= 30
       0  2191.3    19.7 2179.38    59.1 2161.39    98.5 2144.88   108.4 2138.34
   187.2 2106.31     197 2099.88   206.9 2094.95   256.1 2076.17   275.8 2070.21
   285.7 2065.47   295.5 2059.57   374.3 2031.25   384.2 2025.24     394 2020.73
   443.3 2002.57   453.2 1999.46     463 1998.03   532.2 1991.99   561.8 1984.89
   571.5 1984.45   591.5 1985.32   601.3 1986.06   680.3 1996.96   848.2 1999.12
   877.9 2000.78   976.6 2009.14   996.4 2012.49  1095.2 2024.22  1105.1 2026.35
#Mann= 3 , 0 , 0
       0      .1       0   571.5    .045       0   591.5      .1       0
Bank Sta=571.5,591.5
XS Rating Curve= 0 ,0
Exp/Cntr=0.3,0.1

Type RM Length L Ch R = 1 ,9113.2  ,301.3,300,298
XS GIS Cut Line= 3
     1879243.955      272413.904     1879660.762      272766.033
     1880106.728      273084.564
#Sta/Elev= 30
       0 2212.88    29.8 2201.52    49.6    2189     129 2157.04   138.9 2152.04
   148.8 2144.06   158.7 2139.04   238.1 2102.95   257.9 2092.22   327.4 2062.37
   347.2 2052.81   357.2 2046.17   367.1 2041.83   396.8 2030.63   416.7  2025.2
   446.4 2013.92   466.3 2002.56   486.1    1994     496 1990.79   535.6 1984.12
   545.6  1983.8   555.6 1984.15   645.3  1995.3   655.2 1995.78     715 1993.17
   764.9 1993.56   814.7 1994.95   904.4 2001.53   954.2 2007.01  1093.7 2028.26
#Mann= 3 , 0 , 0
       0      .1       0   535.6    .045       0   555.6      .1       0
Bank Sta=535.6,555.6
XS Rating Curve= 0 ,0
Exp/Cntr=0.3,0.1

Type RM Length L Ch R = 1 ,8813.2  ,305.4,300.3,304.6
XS GIS Cut Line= 3
     1879076.206      272690.432       1879526.2      273031.752
     1879991.547       273310.96
#Sta/Elev= 30
       0 2179.73    49.5 2156.69    69.4 2144.07    99.1 2128.82   118.9  2123.4
   138.7 2113.57   148.6 2108.19   188.3 2080.88   227.9 2057.72   267.5 2042.56
   287.4 2039.52   336.9 2024.28   356.7 2016.76   366.6    2011   376.5 2007.25
   426.1 1991.75     436 1990.14   554.8 1984.28   564.8 1983.84   574.8 1984.27
   604.3 1992.25   742.4 1999.32   801.6  2007.2   821.3 2008.32     920 2026.71
   989.1 2042.93  1018.7 2045.77  1058.1 2054.15  1077.9 2055.61  1107.5 2064.18
#Mann= 3 , 0 , 0
       0      .1       0   554.8    .045       0   574.8      .1       0
Bank Sta=554.8,574.8
XS Rating Curve= 0 ,0
Exp/Cntr=0.3,0.1

Type RM Length L Ch R = 1 ,8513.2  ,293.1,299.6,299.1
XS GIS Cut Line= 3
     1878821.142      273005.607     1879316.439      273230.002
     1879745.463      273590.919
#Sta/Elev= 30
       0 2133.12      89 2089.35     178 2050.19   247.2 2026.78   266.9  2017.9
   306.5 2006.16   336.1 2000.45     346 1996.38   365.8 1993.37     435 1987.12
     524 1983.95   533.8 1984.04   553.8 1985.01   642.1 1991.72   720.8 2001.17
     770 2009.17   789.6 2014.04   819.2 2024.56     829  2030.5   848.7 2037.63
   868.3 2046.99   878.2 2050.14   897.8 2052.41   917.5 2061.52     947  2079.4
   976.5 2094.63   996.2 2106.53  1055.2 2132.96  1084.7 2141.42  1104.4  2150.7
#Mann= 3 , 0 , 0
       0      .1       0   533.8    .045       0   553.8      .1       0
Bank Sta=533.8,553.8
XS Rating Curve= 0 ,0
Exp/Cntr=0.3,0.1

Type RM Length L Ch R = 1 ,8213.2  ,295.2,300,305
XS GIS Cut Line= 3
       1878729.3      273123.975     1879148.585      273476.113
     1879570.237      273822.155
#Sta/Elev= 30
       0 2109.77      10 2108.09    19.9  2104.4    79.6 2075.41   149.3 2045.36
   169.2 2040.66     219 2025.03   238.9 2017.13   288.7 2003.06   308.6 1999.95
   338.5 1991.34   358.4 1987.87   537.5 1982.08   557.5 1981.18   577.3 1980.31
     607  1986.6   676.5 1994.61   745.9 2006.18   775.6 2016.41   795.5 2026.73
   805.4 2030.19     855 2044.74   874.8 2046.32   884.7  2050.2   904.6 2064.89
   944.2 2087.28   964.1 2097.69   983.9 2104.75  1013.7 2123.16    1093 2162.24
#Mann= 3 , 0 , 0
       0      .1       0   537.5    .045       0   557.5      .1       0
Bank Sta=537.5,557.5
XS Rating Curve= 0 ,0
Exp/Cntr=0.3,0.1

Type RM Length L Ch R = 1 ,7913.2  ,305.7,301.8,297.8
XS GIS Cut Line= 3
     1878580.332      273250.713      1878924.45      273674.622
     1879268.568      274098.531
#Sta/Elev= 30
       0 2128.74    19.8 2118.51    79.4 2095.27   119.1  2082.1     139  2070.9
   158.8 2065.21   248.2 2032.05   287.9  2020.6   317.7 2007.82   337.5 2001.78
   377.2 1991.84     407 1987.76   436.8 1981.44     536 1976.96     556  1975.4
   565.8 1975.18     675 1981.87     685 1981.81   704.8 1978.36   714.8 1978.76
   784.2 1985.89   804.1 1991.62   843.8 2009.25   863.7 2015.63   893.4 2019.78
   913.3 2020.57   923.2 2023.07   982.8 2050.13  1012.6 2059.42    1092  2090.9
#Mann= 3 , 0 , 0
       0      .1       0     536    .045       0     556      .1       0
Bank Sta=536,556
XS Rating Curve= 0 ,0
Exp/Cntr=0.3,0.1

Type RM Length L Ch R = 1 ,7611.1  ,315.9,307,299
XS GIS Cut Line= 3
     1878324.424       273468.01     1878694.611      273867.271
     1879104.116      274239.484
#Sta/Elev= 30
       0 2095.84    79.2 2092.68    89.1 2093.96   128.7  2087.7   148.5 2082.18
   178.2 2067.42   207.9 2055.68   227.7 2052.93   267.3 2037.84   346.5 2010.47
   366.3 2007.67   455.4 1981.08     495 1975.16   544.5 1964.47   558.5 1963.62
   578.5 1963.38   653.2 1962.46   692.7 1964.87     752 1978.73   791.5 1977.45
   880.4 2000.96   900.2  2007.5   939.8 2011.32   949.6  2014.3   989.2 2030.55
  1008.9  2041.3  1038.6  2053.4  1048.4 2056.88  1058.3 2058.78  1097.9 2073.72
#Mann= 3 , 0 , 0
       0      .1       0   558.5    .045       0   578.5      .1       0
Bank Sta=558.5,578.5
XS Rating Curve= 0 ,0
Exp/Cntr=0.3,0.1

Type RM Length L Ch R = 1 ,7304.2  ,332.3,332.4,331.5
XS GIS Cut Line= 3
      1878009.64      273945.278     1878526.282       274109.88
     1879056.148      274312.715
#Sta/Elev= 30
       0 2011.41    59.2 1997.46   197.2 1986.69   305.6  1973.2   384.5  1970.2
   404.2 1973.34   423.9  1974.1   483.1 1961.16   548.6 1958.34   568.6 1956.35
   572.1  1956.1   701.5 1957.76   721.4 1960.57   751.3 1971.92   761.2 1973.73
   791.1 1973.44     801 1975.28   820.9 1985.17   830.9  1993.4   850.8 2003.63
   860.8 2006.44   880.7 2007.68   900.6 2011.47   920.5 2019.09   990.2 2038.91
    1010 2047.65  1059.8 2063.86  1079.7 2068.54  1089.7 2073.58  1109.6 2080.43
#Mann= 3 , 0 , 0
       0      .1       0   548.6    .045       0   568.6      .1       0
Bank Sta=548.6,568.6
XS Rating Curve= 0 ,0
Exp/Cntr=0.3,0.1

Type RM Length L Ch R = 1 ,6971.7  ,339.5,340,340.6
XS GIS Cut Line= 3
     1877956.362      274169.105     1878473.975      274403.206
     1878967.542      274626.838
#Sta/Elev= 30
       0 2037.88   109.6 2000.95   119.6 1996.02   139.5 1989.53   229.2 1980.61
     309 1975.02   398.7 1956.86   408.6 1955.84   458.5 1952.58   587.8 1949.22
   601.7 1949.69   621.7 1951.23   656.8 1955.82   676.5  1965.5   686.3 1968.84
     706  1971.7   735.6 1979.09   745.4 1981.85   765.1 1990.96   784.8 1996.15
   804.5 1999.94   834.1 2000.33   853.8  2007.8   883.4 2013.14   922.8 2016.76
   932.6 2019.14   981.9 2021.96  1001.6 2027.04  1021.3 2030.26    1110 2025.36
#Mann= 3 , 0 , 0
       0     .06       0   601.7    .045       0   621.7     .06       0
Bank Sta=601.7,621.7
XS Rating Curve= 0 ,0
Exp/Cntr=0.3,0.1

Type RM Length L Ch R = 1 ,6631.7  ,250.6,241,231.4
XS GIS Cut Line= 3
     1877848.162      274321.344     1878106.497      274583.475
     1878768.874      274868.235
#Sta/Elev= 30
       0 2040.68    59.7 2025.53    89.5 2021.71   119.4 2021.49   208.9 2013.28
   268.6 2013.23   288.5 2011.62   338.2 2001.13   437.2 1969.52   506.3 1954.27
   526.1  1947.9   535.9  1947.3   536.9  1947.3   556.9 1947.63     694 1954.47
   713.7 1957.43   733.5 1963.38   743.4 1965.07   753.2  1965.2   792.7 1961.04
   802.6 1961.45   842.1 1964.08   901.4 1972.02   921.1 1976.72   950.8 1986.53
   980.4 1989.91  1000.1 1994.54  1039.6 2006.83  1059.4 2016.19    1089 2022.44
#Mann= 3 , 0 , 0
       0      .1       0   536.9    .045       0   556.9      .1       0
Bank Sta=536.9,556.9
XS Rating Curve= 0 ,0
Exp/Cntr=0.3,0.1

Type RM Length L Ch R = 1 ,6390.7  ,275.6,281.9,288.1
XS GIS Cut Line= 3
     1877718.065      274670.049     1878067.807      274886.806
     1878831.643      274908.972
#Sta/Elev= 30
       0 2018.76    58.8 2018.25   127.4 2019.93   215.5 2017.69   284.1 2005.78
   323.3 1993.21   342.9 1984.75   372.3 1978.17   431.3 1968.57   441.2 1965.44
   451.2 1963.94   520.6 1954.14   582.3 1947.54   590.1 1947.22   602.3  1947.3
   669.5 1951.13   699.3 1959.77   709.2 1961.47   719.1 1961.08     729 1958.44
     739 1954.06   758.8 1952.22   818.4 1968.81   907.7 1982.35   987.1 2003.61
  1006.9 2010.33  1066.5 2022.76  1086.3 2029.32  1106.2 2034.12  1175.6    2044
#Mann= 3 , 0 , 0
       0      .1       0   582.3    .045       0   602.3      .1       0
Bank Sta=582.3,602.3
XS Rating Curve= 0 ,0
Exp/Cntr=0.3,0.1

Type RM Length L Ch R = 1 ,6108.8  ,347.3,402,435
XS GIS Cut Line= 3
     1877710.448      274729.094     1878012.093      275064.781
     1878828.637      275289.565
#Sta/Elev= 30
       0 2026.56   137.4 2021.37   225.6 2023.84   274.7 2020.22   323.8 2013.39
   353.2  2007.5   431.7 1984.74   441.5 1981.31   461.3 1970.91   550.9 1954.44
   580.8 1950.75   600.8  1949.7   670.5 1956.43   750.2 1948.05     778 1946.77
   780.1 1946.74     798 1948.65   839.9  1954.6   859.8 1958.87   869.8 1959.34
   889.7 1968.17   969.4 1988.06  1039.2 1998.18  1049.1 2001.53  1118.9 2015.52
  1138.8 2021.81  1198.6 2031.71  1218.5 2036.99  1288.3 2049.55  1298.2 2052.86
#Mann= 3 , 0 , 0
       0      .1       0     778    .045       0     798      .1       0
#XS Ineff= 2 , 0
          671.22  1956.2
Permanent Ineff=
       F       F
Bank Sta=778,798
XS Rating Curve= 0 ,0
Exp/Cntr=0.3,0.1

Type RM Length L Ch R = 1 ,5706.8  ,248.7,223.5,219.6
XS GIS Cut Line= 3
     1877662.424      274763.305     1878058.522       275123.59
     1878132.807      275826.204
#Sta/Elev= 30
       0 2023.92    89.2 2019.88   138.8 2020.24   208.2 2023.77   257.8 2022.58
   386.7 2006.13   436.3 1990.54     476 1971.46   485.9 1968.51   525.5 1961.32
   585.2 1953.02   595.2 1953.14     635 1957.78   644.9 1956.36   664.8 1949.16
   674.8 1947.57     723  1946.3     743 1946.35   794.2 1946.72   843.9 1952.25
   873.8 1959.38   913.6  1966.8   933.5 1968.74  1003.2    1987    1023 1989.84
  1072.8 2001.69  1112.6 2009.19  1122.6 2009.32  1172.3 2016.36    1242 2018.66
#Mann= 3 , 0 , 0
       0      .1       0     723    .045       0     743      .1       0
#XS Ineff= 2 , 0
          636.46  1958.1
Permanent Ineff=
       F       F
Bank Sta=723,743
XS Rating Curve= 0 ,0
Exp/Cntr=0.3,0.1

Type RM Length L Ch R = 1 ,5483.3  ,342.2,327.2,316.1
XS GIS Cut Line= 3
     1877601.064      274782.685     1877860.428      275131.328
     1877955.143      275868.606
#Sta/Elev= 30
       0 2019.45    69.1 2017.92   118.5 2011.93   138.3 2011.22   227.1 2016.21
   296.3 2017.09   325.9 2015.66   414.8 1996.47   424.7  1997.1   434.5 1995.45
   474.2 1983.71   503.9 1976.53   543.6 1971.38   553.5 1967.11   573.3 1951.47
   583.2 1947.42   588.7 1946.94   593.1 1946.56   608.7 1948.15   672.4 1952.38
   692.2 1954.49     712 1958.55     722 1958.67   811.2 1980.64   821.1 1980.72
   880.5 1999.15   900.4 2003.82   989.6 2010.65  1118.4 2010.75  1177.9 2014.06
#Mann= 3 , 0 , 0
       0      .1       0   588.7    .045       0   608.7      .1       0
Bank Sta=588.7,608.7
XS Rating Curve= 0 ,0
Exp/Cntr=0.3,0.1

Type RM Length L Ch R = 1 ,5156    ,303.6,299.7,290.5
XS GIS Cut Line= 3
     1877242.124      274972.373      1877583.26       275388.05
     1877877.709      275901.972
#Sta/Elev= 30
       0  2012.2   139.4 2012.08   209.1 2007.09   298.7 1994.43   328.6 1987.56
   338.6 1984.74   358.5 1974.99   398.3 1958.33   418.2 1951.68   438.2 1950.74
     468  1953.1   497.9 1948.15   507.9 1946.32   527.7  1947.9   567.4 1950.63
   577.2 1952.34   606.8 1959.96   626.6 1966.93   675.9 1978.91   705.6 1990.18
   725.3 1993.24   784.5  1997.6   804.3 2000.73     824 2002.13   912.9 2002.22
     982 2000.23  1031.3 2000.22  1060.9 2002.88  1100.4 2009.31    1130 2011.68
#Mann= 3 , 0 , 0
       0      .1       0   497.9    .045       0   527.7      .1       0
#XS Ineff= 2 , 0
           468.1  1953.1
Permanent Ineff=
       F       F
Bank Sta=497.9,527.7
XS Rating Curve= 0 ,0
Exp/Cntr=0.3,0.1

Type RM Length L Ch R = 1 ,4856    ,342.7,331.5,321.8
XS GIS Cut Line= 3
     1876986.086      275248.474     1877392.556      275618.515
     1877816.041      275963.694
#Sta/Elev= 30
       0 1973.28      90 1979.22   109.9 1982.27   199.9 1989.34   229.9 1995.14
   239.9 1996.05   339.8 1999.07   349.8 1996.22   369.8 1987.15   409.8 1955.72
   419.8 1952.44   479.7 1947.43   539.7 1944.11   559.7 1945.87   589.4 1948.41
   599.4 1950.37   639.1 1965.27     649 1966.63     659 1966.09   678.8 1960.66
   688.8  1961.3   718.6 1970.25   768.2 1987.65     798 1993.94   877.5 1998.92
     957 2006.02   976.8 2005.68  1006.6 2007.08  1066.2 2004.01    1096 2003.72
#Mann= 3 , 0 , 0
       0      .1       0   539.7    .045       0   559.7      .1       0
Bank Sta=539.7,559.7
XS Rating Curve= 0 ,0
Exp/Cntr=0.3,0.1

Type RM Length L Ch R = 1 ,4524.2  ,273.9,274.6,275.4
XS GIS Cut Line= 3
     1876690.436      275691.562     1877345.074       275912.87
     1877671.666      276132.293
#Sta/Elev= 30
       0 1993.87    39.5 1990.99      79 1990.08     158  1994.7   217.2 1993.27
   236.9 1988.94   246.8 1981.69   286.3 1959.27     306 1949.47   315.9 1946.36
   325.8 1945.08   365.3 1945.29   404.8 1943.57   454.1 1951.51     464 1950.78
   483.7 1944.79   498.6 1945.47   552.8 1952.88   592.3 1961.48   641.7 1968.68
   661.4 1973.96   700.9 1992.38   740.2 2000.02   818.9 2001.98   838.6 2000.93
   917.3 1988.08   956.6 1983.61   986.1 1985.49    1055  1996.8  1084.5 1997.08
#Mann= 3 , 0 , 0
       0      .1       0   483.7    .045       0   498.6      .1       0
#XS Ineff= 2 , 0
          454.13 1951.52
Permanent Ineff=
       F       F
Bank Sta=483.7,498.6
XS Rating Curve= 0 ,0
Exp/Cntr=0.3,0.1

Type RM Length L Ch R = 1 ,4249.7  ,201.7,199.8,197.9
XS GIS Cut Line= 3
     1876580.502      275938.117     1877096.678      276116.101
     1877612.853      276294.086
#Sta/Elev= 30
       0 2016.45     9.9 2014.36    39.7 2005.75    79.4 1997.84   198.6 1985.94
   238.2 1970.12   258.1 1963.15   297.8 1955.72   357.4 1949.13   377.2 1945.39
   387.2 1944.42   446.7 1941.57   456.6    1942   486.4 1949.43   496.4 1950.03
   525.8 1943.18   536.1 1943.89   545.8 1949.74   575.8 1959.11   615.5 1969.49
   635.4 1977.51   655.2 1982.78   665.1 1984.49     675 1985.14   694.9 1984.38
   843.8 1971.17   873.6 1972.97   982.8 1986.26  1032.4 1988.16    1092 1987.34
#Mann= 3 , 0 , 0
       0      .1       0   525.8    .045       0   545.8      .1       0
Bank Sta=525.8,545.8
XS Rating Curve= 0 ,0
Exp/Cntr=0.3,0.1

Type RM Length L Ch R = 1 ,4049.8  ,285.9,285,284.1
XS GIS Cut Line= 3
     1876462.881      276137.206     1876986.134      276292.922
     1877514.843      276430.782
#Sta/Elev= 30
       0 2060.24    59.6 2048.97    79.4 2042.64   148.9 2028.93   158.8 2024.44
   228.3 2008.34   277.9 1994.04   317.6 1980.16   327.6  1972.9   347.4 1967.68
   476.4 1946.76   496.3 1945.11   555.9 1948.34   565.8 1947.04   575.7 1942.22
   585.7 1940.86     589 1941.33   595.6 1942.26     609 1947.48   625.4 1954.16
   635.3 1956.65     695 1965.11   724.8 1964.55   774.4 1959.26   814.2 1956.43
   863.8  1956.3  1012.8  1959.6  1032.7 1961.21  1072.4 1968.38  1092.3 1969.89
#Mann= 3 , 0 , 0
       0      .1       0     589    .045       0     609      .1       0
Bank Sta=589,609
XS Rating Curve= 0 ,0
Exp/Cntr=0.3,0.1

Type RM Length L Ch R = 1 ,3764.8  ,412.6,414.8,417.1
XS GIS Cut Line= 3
     1876397.524      276455.486      1876930.78       276572.76
     1877464.037      276690.034
#Sta/Elev= 30
       0  2053.8   158.8 2030.86   287.9 2015.95   307.8  2012.2   317.7 2008.79
   337.5 2006.04   387.2 2001.76   426.9 2000.44   436.8 1998.46   466.6  1983.8
   486.4 1968.82   516.2 1952.51   526.2 1949.21     546 1945.91   564.2 1939.18
   565.8 1938.61   584.2 1940.83   615.5 1951.28   625.4 1952.26   665.1 1951.28
     685  1952.7   714.8 1959.91   724.7 1965.23   744.6 1970.44   794.2 1978.95
     814 1983.75   843.8 1986.85   992.7 1996.81  1042.4  1995.5    1092 1990.27
#Mann= 3 , 0 , 0
       0      .1       0   564.2    .045       0   584.2      .1       0
Bank Sta=564.2,584.2
XS Rating Curve= 0 ,0
Exp/Cntr=0.3,0.1

Type RM Length L Ch R = 1 ,3349.9  ,239.4,237.6,235.8
XS GIS Cut Line= 3
     1876352.526      276822.317     1876873.258      276986.492
     1877393.991      277150.667
#Sta/Elev= 30
       0 2012.84    39.7 2012.77    59.6 2009.28   119.1  1992.5     129 1986.93
   158.8 1976.44   198.6 1970.09   218.4 1960.72   248.2 1949.89     268 1945.39
     407 1941.21   436.8 1941.58   476.5 1945.28   513.3 1936.78   526.2 1936.13
   533.3 1936.88     546 1939.22   565.8 1945.89   605.6 1954.89   625.4  1960.8
   635.4 1965.06   645.3 1971.72     685 1989.92   694.9 1994.29   704.8 1997.12
   714.8    1998   774.3 1997.28   903.4 1994.14  1032.4 1994.63    1092 1992.17
#Mann= 3 , 0 , 0
       0      .1       0   513.3    .045       0   533.3      .1       0
#XS Ineff= 2 , 0
          474.79 1945.77
Permanent Ineff=
       F       F
Bank Sta=513.3,533.3
XS Rating Curve= 0 ,0
Exp/Cntr=0.3,0.1

Type RM Length L Ch R = 1 ,3112.3  ,221.6,221.5,221.3
XS GIS Cut Line= 3
     1876251.978      277083.596     1876783.942      277207.633
     1877315.349      277334.603
#Sta/Elev= 30
       0 1985.14    99.3  1989.6   129.1 1988.76   158.9 1984.28   168.8  1983.9
   228.4 1987.78   248.3 1982.45   268.2 1974.64     298  1961.2   327.7 1946.08
   377.4 1937.28   456.8 1936.88   466.8  1937.6   486.6 1942.74   496.6 1943.33
   516.4 1941.66   551.8 1935.38   556.2 1934.78   571.8 1936.36   625.7 1948.02
   635.6 1951.06   655.5 1960.14     725 1982.04     735 1987.86   754.8    1992
   834.3 1999.25   913.8 2003.48   993.3 2011.73  1062.8  2014.5  1092.6 2017.13
#Mann= 3 , 0 , 0
       0      .1       0   551.8    .045       0   571.8      .1       0
#XS Ineff= 2 , 0
           496.2 1943.16
Permanent Ineff=
       F       F
Bank Sta=551.8,571.8
XS Rating Curve= 0 ,0
Exp/Cntr=0.3,0.1

Type RM Length L Ch R = 1 ,2890.7  ,193.4,193.3,193.2
XS GIS Cut Line= 2
     1876306.629      277324.289     1877060.314      277499.169
#Sta/Elev= 30
       0 1968.36    19.8 1966.03    29.8    1963    59.5 1958.29   109.1  1948.9
     129 1946.87   198.4 1941.37   238.1 1940.46   277.7  1936.9   347.2 1936.89
     367 1940.42   376.9 1941.06   386.8 1940.44   426.5 1935.39   438.5 1933.28
   446.4 1932.15   456.3 1932.02   458.5 1932.28   466.2 1933.18     486  1938.3
     496 1940.32   515.8 1943.49   525.7 1946.26   595.2 1961.18   605.1 1965.62
   674.5 1980.99   684.4  1984.2   694.4 1986.65   753.9 1998.76   773.7 2005.82
#Mann= 3 , 0 , 0
       0      .1       0   438.5    .045       0   458.5      .1       0
#XS Ineff= 2 , 0
          377.35  1940.8
Permanent Ineff=
       F       F
Bank Sta=438.5,458.5
XS Rating Curve= 0 ,0
Exp/Cntr=0.3,0.1

Type RM Length L Ch R = 1 ,2697.4  ,245.7,248.3,251.7
XS GIS Cut Line= 3
     1876142.377      277487.115      1876674.77       277608.25
     1877207.163      277729.385
#Sta/Elev= 30
       0 1999.75    39.7 2000.93   158.8 1997.41   208.5 1997.66   218.4 1995.48
     278 1972.14   287.9 1965.99   297.8 1961.57   347.4 1946.61   377.2 1939.11
   456.6 1932.66   466.6 1933.52   486.4 1938.15   506.3 1939.09   526.2  1936.6
   560.3 1930.32   575.8 1929.68   580.3 1930.19   635.4 1940.24     685 1942.74
   724.7  1946.8   774.3 1956.33   784.2 1960.32   853.8 1973.68   863.7 1977.37
   933.2 1994.87     953 2003.59  1012.6 2022.02  1032.4 2031.54    1092  2047.6
#Mann= 3 , 0 , 0
       0      .1       0   560.3    .045       0   580.3      .1       0
#XS Ineff= 2 , 0
          497.13 1939.11
Permanent Ineff=
       F       F
Bank Sta=560.3,580.3
XS Rating Curve= 0 ,0
Exp/Cntr=0.3,0.1

Type RM Length L Ch R = 1 ,2449    ,300.7,299.9,298.2
XS GIS Cut Line= 3
     1876124.061       277680.66     1876643.325      277855.133
     1877154.056      278047.291
#Sta/Elev= 30
       0 1997.37   159.4 1980.24   219.1 1970.98   298.8 1946.74   318.7 1938.75
   328.7 1936.62   378.5 1933.07   408.4  1926.7   418.3 1925.87   428.3 1927.19
   448.2 1933.85   468.1 1937.71   478.1 1936.96     488 1933.45   517.9 1926.63
   537.8  1924.8   557.8 1927.29   577.6 1931.81   627.2 1938.79   696.6 1943.47
   815.7  1966.5   865.3  1963.6   875.2 1963.89     895 1966.77   914.9  1972.4
   924.8 1979.09   994.3 2006.53  1014.1 2016.94  1083.6 2037.74  1093.5 2043.18
#Mann= 3 , 0 , 0
       0      .1       0   537.8    .045       0   557.8      .1       0
#XS Ineff= 2 , 0
           469.2 1937.18
Permanent Ineff=
       F       F
Bank Sta=537.8,557.8
XS Rating Curve= 0 ,0
Exp/Cntr=0.3,0.1

Type RM Length L Ch R = 1 ,2149    ,307.6,299.8,291.4
XS GIS Cut Line= 3
     1876002.494      277971.759     1876524.053       278129.29
     1877053.318      278288.291
#Sta/Elev= 30
       0 1976.97   118.9 1973.78   178.3 1973.25   257.6 1966.88   267.5 1965.75
   277.4 1963.28   287.3 1958.14   346.7 1939.11   366.5 1934.32   406.2 1933.23
   505.2 1934.92   515.1 1933.06     525 1929.58   534.8 1922.83   544.8 1920.71
   554.8 1921.09   663.2 1936.56   702.7 1939.65   771.8 1963.99   791.5 1974.25
   821.2 1984.07   840.9 1988.76   870.5 1993.19   939.6 1997.17   959.3 1999.36
  1008.6 2001.53  1018.5  2002.8  1028.4 2005.16  1038.2 2010.63  1097.5 2026.33
#Mann= 3 , 0 , 0
       0      .1       0   534.8    .045       0   554.8      .1       0
Bank Sta=534.8,554.8
XS Rating Curve= 0 ,0
Exp/Cntr=0.3,0.1

Type RM Length L Ch R = 1 ,1849    ,271.6,279.2,287.6
XS GIS Cut Line= 3
     1875934.471      278442.627     1876495.354      278414.091
     1877041.499      278373.549
#Sta/Elev= 30
       0 2049.73    39.4 2035.52    98.5  2021.2   118.2 2014.22   177.4 2000.42
   256.2 1973.25   275.9 1963.81   325.1 1950.57   354.7 1943.98   413.8 1937.76
   433.5 1934.47   453.2 1932.64   482.8 1933.47   502.5  1931.2   522.2  1926.1
   541.9  1918.8   551.6 1918.75   571.6 1920.92   591.5 1924.37   661.2 1932.38
     691 1933.31   740.8 1948.38   760.8 1957.16   840.4 1977.82   860.3 1979.58
   959.9 1982.97  1029.6 1988.85  1059.5 1994.77  1079.4 2002.73  1109.3  2011.8
#Mann= 3 , 0 , 0
       0      .1       0   551.6    .045       0   571.6      .1       0
Bank Sta=551.6,571.6
XS Rating Curve= 0 ,0
Exp/Cntr=0.3,0.1

Type RM Length L Ch R = 1 ,1569.9  ,347.5,346.5,345.5
XS GIS Cut Line= 3
     1875920.803      278530.008      1876538.77      278707.851
     1876988.968      278775.624
#Sta/Elev= 30
       0 2048.58    39.6 2038.67    59.4 2031.55   128.6 2013.98   138.5 2009.71
   207.8 1994.24   227.5 1986.51   296.8 1968.87   306.7 1963.94   375.9 1946.02
   395.7 1935.99   405.6 1933.27   415.5 1931.94   474.9 1932.28   541.9 1919.66
     554 1916.52   561.9 1916.38   563.9 1916.35   623.3 1928.07   692.5 1933.14
   751.9 1943.11   791.5 1952.98   801.4 1957.19   811.3 1959.49   870.7 1969.64
   900.4 1978.13   949.9 1989.51   969.7  1996.1  1048.8 2015.33  1098.3 2024.15
#Mann= 3 , 0 , 0
       0      .1       0   541.9    .045       0   561.9      .1       0
Bank Sta=541.9,561.9
XS Rating Curve= 0 ,0
Exp/Cntr=0.3,0.1

Type RM Length L Ch R = 1 ,1223.3  ,153.3,155,156.6
XS GIS Cut Line= 3
     1875873.299      278888.921     1876148.773      278961.658
     1876919.472      279152.502
#Sta/Elev= 30
       0 2002.27    49.1 1989.24   108.1 1978.46   117.9 1975.12   147.4 1969.06
   245.6 1957.21   265.3 1952.08   284.9 1939.45   314.7 1931.28   433.8 1930.01
   473.5 1930.89   503.3  1924.7     533  1915.8   540.3 1916.17   560.3 1919.61
   582.7    1923   602.5 1919.67   612.4  1916.1   622.4 1916.39   681.9 1921.47
   781.2    1938   810.9    1941   850.6 1954.08   860.6 1960.36   900.2 1972.88
     930 1980.17   949.9 1987.46  1029.3 2004.33    1059 2009.15  1078.9 2014.41
#Mann= 3 , 0 , 0
       0      .1       0   540.3    .045       0   560.3      .1       0
#XS Ineff= 2 , 0
                          583.71         1922.82
Permanent Ineff=
       F       F
Bank Sta=540.3,560.3
XS Rating Curve= 0 ,0
Exp/Cntr=0.3,0.1
